HEC-RAS study MFWILLIAMSRV.prj: MFWILLIAMSRV

--- MFWILLIAMSRV.g01 (geometry) --- (continued)

Type RM Length L Ch R = 1 ,23006   ,266.1,298.3,310.2
XS GIS Cut Line= 3
2168786.69705806478083.4930274622168835.71394038478549.153409526
2169183.28819685478785.325660717
#Sta/Elev= 30
       0 3126.74    25.8 3119.17    57.5 3106.44    78.1 3091.61    86.2 3087.88
   110.3 3068.73   138.4 3055.47   226.9 3029.96   263.1 3012.27   283.2 3009.79
   319.4 3009.47   335.5  3004.4   379.8 3002.17   387.8 3002.97   403.9 3009.13
   432.1 3009.82   460.2  3006.5   483.3  3010.7   517.2 3006.08   549.2 3006.89
   566.43003.565   601.53003.646     632 3004.59   647.7 3012.99   674.7 3018.44
   696.1 3029.34   739.6 3057.75   807.3 3076.53   821.8 3077.91   888.5 3101.17
#Mann= 5 ,-1,0
       0      .1       0   566.4    .045       0   601.5      .1       0
  658.23     .06       0  728.23      .1       0
#XS Ineff= 2 , 0
          542.03 3031.36
Permanent Ineff=
       F       F
Bank Sta=566.4,601.5
XS Rating Curve= 0 ,0
Exp/Cntr(USF)=0,0
Exp/Cntr=0.3,0.1

Type RM Length L Ch R = 1 ,22707   ,397.5,411.4,421
XS GIS Cut Line= 3
2168752.37073314478099.4657270212168748.61297937478457.819983167
2168703.10980449478920.481204584
#Sta/Elev= 30
       0 3122.04    41.7 3106.86    77.1  3085.6    89.7 3073.27   105.7 3065.04
   177.7 3037.18   229.7 3027.16   257.7 3012.29   306.7 3005.53   325.7 3000.74
   353.7 2999.05   369.8 3002.98   397.9 3002.34     422  3006.5     482 3004.31
   530.6 3005.94   556.12993.971   570.4 2991.56   587.42992.906   635.1 2996.02
   639.1 2997.18   651.1 3006.32   667.2 3010.09   679.3 3019.97   703.4 3051.24
   731.5 3077.19   763.7 3095.51   779.8 3099.34   795.8 3110.64   823.3 3120.17
#Mann= 4 ,-1,0
       0      .1       0   556.1    .045       0   587.4     .06       0
  758.37      .1       0
Bank Sta=556.1,587.4
XS Rating Curve= 0 ,0
Exp/Cntr(USF)=0,0
Exp/Cntr=0.3,0.1

Type RM Length L Ch R = 1 ,22296   ,367.3,361.7,353.1
XS GIS Cut Line= 3
2168657.49783352 478081.220938632168259.76144661478654.107294086
2168257.93696777478836.555177989
#Sta/Elev= 30
       0  3125.4    19.4 3116.71      34 3113.15    58.4 3101.16   189.9 3049.55
   233.7 3018.44   243.4 3014.64   268.8 2999.13   311.6 2994.05   345.7 2993.47
   374.9 2995.87   381.1 2993.89   402.1 2981.11   462.6 2980.54   501.5 2979.57
   506.4 2980.96   516.1 2985.22     521 2985.62   540.5 2980.76   550.2 2980.84
   574.6 2987.37   584.3  2993.7   590.1 2995.17   624.6 2994.34   654.6 2997.59
   676.8 2995.58   693.6 2999.86   728.5 3022.68   752.5 3035.48   879.9 3093.91
#Mann= 5 ,-1,0
       0      .1       0   462.6    .045       0   506.4      .1       0
     530     .06       0  707.42      .1       0
#XS Ineff= 1 ,-1
  518.72879.8759 3001.65
Permanent Ineff=
       F
Bank Sta=462.6,506.4
XS Rating Curve= 0 ,0
Exp/Cntr(USF)=0,0
Exp/Cntr=0.3,0.1

Type RM Length L Ch R = 1 ,21934   ,573.7,551,519
XS GIS Cut Line= 4
 2168002.5359731478011.7622830292168074.61590863478300.776409349
2168044.73161727478390.7365342032168053.72379752478804.099938039
#Sta/Elev= 30
       0 3134.18    26.2 3122.53    38.6 3115.02    59.2 3111.14   108.6 3078.28
   170.5 3040.56   203.5 3016.91   224.1 2997.48   244.7 2984.22   256.6 2979.24
     290 2972.96   310.9 2973.28   323.6 2969.45   327.8  2967.6   347.6 2967.43
   364.1 2969.77   374.2 2976.39   443.1  2975.8   463.1 2982.05   471.1 2979.34
   495.1 2978.62   511.1 2988.17   519.1 2989.91   603.2 2988.44   631.2 2990.69
   651.2  3000.3   680.4  3018.9   707.2  3038.9   771.2 3066.67   806.1 3077.45
#Mann= 5 ,-1,0
       0      .1       0   323.6    .045       0   364.1      .1       0
  367.87     .06       0  562.66      .1       0
Bank Sta=323.6,364.1
XS Rating Curve= 0 ,0
Exp/Cntr(USF)=0,0
Exp/Cntr=0.3,0.1

Type RM Length L Ch R = 1 ,21383   ,326.6,380,407.7
XS GIS Cut Line= 3
2167556.28512728478296.3549391272167668.98191056478585.351395534
2167947.77556513 478832.90622031
#Sta/Elev= 30
       0 3072.66    30.9 3049.47    35.2 3042.91    46.9 3017.21    52.4 3009.78
      61 3002.25    98.8  2975.2     121 2965.21   159.7 2961.45   176.9 2955.96
   189.8 2958.41   207.5 2958.74   228.4 2954.85   252.9 2959.19   288.5 2960.62
   312.3 2960.64   325.2 2957.75     368 2956.51   374.7 2957.56   388.2 2965.93
   411.5 2967.06   436.4 2982.55   454.5 2989.95   465.3 2992.39   484.6 3002.45
   496.5 3005.37   508.7 3011.72   533.3 3021.29   587.1 3037.95     683  3073.7
#Mann= 5 ,-1,0
       0      .1       0   325.2    .045       0   374.7      .1       0
  420.19     .06       0  570.19      .1       0
#XS Ineff= 2 , 0
          290.57 2983.37
Permanent Ineff=
       F       F
Bank Sta=325.2,374.7
XS Rating Curve= 0 ,0
Exp/Cntr(USF)=0,0
Exp/Cntr=0.3,0.1

Type RM Length L Ch R = 1 ,21003   ,386.8,381.1,365.4
XS GIS Cut Line= 4
2167362.70982505  478329.88994242167389.87041955 478605.18141324
2167294.04621631478811.8335638942167405.62238771479102.698211842
#Sta/Elev= 30
       0 3093.89    26.3 3082.46    35.5 3076.55    55.5 3072.91    75.7  3061.1
    87.7 3057.19   117.8 3041.35   126.9 3029.57   140.3 3007.21     152 2985.27
     156 2980.74   208.3 2951.74   224.4 2948.16   298.7 2952.51   319.32948.007
   333.9 2946.69   376.32947.943   391.3  2954.8   404.5 2953.06   448.6 2956.58
   479.4 2955.86   514.4 2959.16   540.1 2956.05   553.6 2962.37   587.3 2969.71
   610.9 2981.23   644.4 3002.18   722.6 3063.22   770.3 3070.44   815.9 3091.23
#Mann= 4 ,-1,0
       0      .1       0   319.3    .045       0   376.3     .06       0
  554.42      .1       0
#XS Ineff= 2 , 0
          296.62 2970.44
Permanent Ineff=
       F       F
Bank Sta=319.3,376.3
XS Rating Curve= 0 ,0
Exp/Cntr(USF)=0,0
Exp/Cntr=0.3,0.1

Type RM Length L Ch R = 1 ,20622   ,283.8,311.7,320.4
XS GIS Cut Line= 3
 2167039.1851033478269.1422590512167004.52000535478809.187995403
2166750.91744673478940.550471813
#Sta/Elev= 30
       0 3064.72    12.1 3063.05    60.2 3045.14   156.4  3000.7   200.4 2983.83
   240.5 2950.78   256.6 2942.64   300.7 2937.62   332.7 2940.46   343.8 2939.11
   380.8  2937.6   390.8 2939.22   400.9  2946.5   420.9 2950.08   458.6 2952.59
   469.9 2950.09     485 2950.97     493 2954.44   526.4 2956.85   541.1 2961.03
   559.2 2956.38   631.6  2959.6   663.1 2957.75   717.2 2958.89   726.2 2962.65
   749.1 2979.98   766.9 3005.67   771.3 3009.18   789.3 3019.75   826.8  3034.4
#Mann= 4 ,-1,0
       0      .1       0   343.8    .045       0   390.8     .06       0
     490      .1       0
#XS Ineff= 2 , 0
          270.67 2952.94
Permanent Ineff=
       F       F
Bank Sta=343.8,390.8
XS Rating Curve= 0 ,0
Exp/Cntr(USF)=0,0
Exp/Cntr=0.3,0.1

Type RM Length L Ch R = 1 ,20311   ,416.2,445.5,462.4
XS GIS Cut Line= 3
2166994.31960208478201.7146703792166657.86902594478628.564590339
2166526.50654953478734.384363003
#Sta/Elev= 30
       0 3068.72    26.8 3061.67    55.2 3048.33    80.8 3029.52   100.8 3008.28
   126.6 2986.68   154.9 2965.11   167.4 2956.57     192 2944.88   214.8 2938.08
   254.6 2937.01   308.8 2939.89   320.2 2938.38   330.4 2932.59   365.3 2930.37
   374.3 2928.77   405.6  2930.4   428.4 2934.54   447.5 2935.72   482.5 2935.08
   502.4 2937.18   518.8 2935.76   545.7 2938.71     556 2944.83   582.7 2966.46
   596.4 2973.88   617.6 2991.39   648.4 3010.34   697.5 3030.64   712.2 3034.91
#Mann= 5 ,-1,0
       0      .1       0     350     .06       0   365.3    .045       0
   405.6     .06       0     510      .1       0
Bank Sta=365.3,405.6
XS Rating Curve= 0 ,0
Exp/Cntr(USF)=0,0
Exp/Cntr=0.3,0.1

Type RM Length L Ch R = 1 ,19865   ,379.6,357.1,332.8
XS GIS Cut Line= 4
2166825.63894064  477985.27302332166649.37754945478138.320795568
 2166420.2799943 478113.268377152166256.07689879 478332.67820662
#Sta/Elev= 30
       0 3062.58    20.8 3060.82    42.6 3051.29    66.2 3036.11    86.7 3019.71
   100.2 2993.83     103 2989.93   108.7  2984.5   155.6 2947.74   176.8 2935.53
   192.6 2928.29   207.3 2924.31   219.1 2923.01   262.8 2923.56   286.3 2918.08
     303 2914.47   317.5 2918.17   347.3 2925.01   387.6 2927.31   447.9 2922.25
   468.8 2923.34   483.9 2922.59   506.8 2924.35   517.5 2928.26   553.7 2947.67
   578.7  2955.8   592.5 2958.16     651 2974.66   673.6 2982.72   737.9 3008.81
#Mann= 4 ,-1,0
       0      .1       0   286.3    .045       0   317.5     .06       0
  403.43      .1       0
Bank Sta=286.3,317.5
XS Rating Curve= 0 ,0
Exp/Cntr(USF)=0,0
Exp/Cntr=0.3,0.1

Type RM Length L Ch R = 1 ,19508   ,435.2,441.6,443.1
XS GIS Cut Line= 4
2166531.76838442477697.6632741942166393.84689439477900.295352055
2166337.52209937478128.3420831062166250.26554893478306.279479224
#Sta/Elev= 30
       0 3040.65    18.8 3033.43    33.3 3018.46    47.8 3008.81      80 2981.73
     101 2962.49   117.4 2950.28   134.9 2939.34   155.7 2919.93   169.52910.221
   186.5 2908.94   206.2  2910.2   241.3 2914.62   274.9 2910.62   296.8 2911.78
   353.2 2910.04   357.3  2911.4   361.4 2914.79   369.6 2917.21   431.4 2919.14
   455.4 2921.77   472.6 2922.04   484.6  2926.4   503.2    2939     521 2947.83
   583.4 2966.12   614.6 2978.11   623.5 2979.37     655 2993.79   678.2 3001.67
#Mann= 5 ,-1,0
       0      .1       0   169.5    .045       0   206.2      .1       0
     210     .06       0  315.12      .1       0
#XS Ineff= 1 ,-1
  240.03   664.5 2929.32
Permanent Ineff=
       F
Bank Sta=169.5,206.2
XS Rating Curve= 0 ,0
Exp/Cntr(USF)=0,0
Exp/Cntr=0.3,0.1

Type RM Length L Ch R = 1 ,19066   ,400.4,390.1,377.9
XS GIS Cut Line= 3
2166224.54439272  477573.03312472165951.48449707477915.951585307
2165884.75125889478087.387892858
#Sta/Elev= 30
       0 3015.55     6.1 3013.56    37.4 2997.07      82  2979.2   112.7 2965.03
   122.6 2958.55   133.1  2948.8   154.7 2932.54     174 2919.32   182.5 2915.63
   196.8 2911.87   214.9  2901.5   225.3 2899.81     261 2901.97   289.6 2900.34
   322.3 2901.36   344.8 2896.83     373 2895.22   387.5 2896.57   404.1 2897.19
   424.6 2902.98   452.5 2903.55   469.7  2906.8   478.3 2913.14   488.2 2922.92
   512.6 2943.83   522.2 2949.18   546.9 2969.13   555.6 2974.66   622.3 3003.08
#Mann= 4 ,-1,0
       0      .1       0   344.8    .045       0   387.5     .06       0
  498.35      .1       0
Bank Sta=344.8,387.5
XS Rating Curve= 0 ,0
Exp/Cntr(USF)=0,0
Exp/Cntr=0.3,0.1

Type RM Length L Ch R = 1 ,18676   ,434.5,454,473
XS GIS Cut Line= 3
2165757.06767073477409.8181541552165683.91519168477518.881850195
2165626.72325352477976.417355531
#Sta/Elev= 30
       0 3005.46    13.7 3002.26    23.1 2996.32    37.8 2990.32    63.6 2975.81
    87.8 2958.82    98.2 2948.29     104 2944.28   121.3 2940.58   141.7  2927.8
   165.4 2917.17   197.6 2912.18   206.2 2909.49   218.3 2902.55   234.4 2897.55
   242.5 2891.06     255 2886.33   262.6 2884.44   270.7 2884.21   283.6 2885.32
   339.2 2885.93   363.4 2888.86   379.5 2898.43   395.7 2899.01   407.8 2907.45
   460.2  2933.4   512.6 2949.49   560.9 2968.96   576.5 2976.34   592.4 2981.75
#Mann= 5 ,-1,0
       0      .1       0     255    .045       0   283.6      .1       0
  291.32     .06       0  391.32      .1       0
Bank Sta=255,283.6
XS Rating Curve= 0 ,0
Exp/Cntr(USF)=0,0
Exp/Cntr=0.3,0.1

Type RM Length L Ch R = 1 ,18222   ,487.6,464,435.3
XS GIS Cut Line= 4
2165441.84698828477409.8181541552165393.96536563477544.152706594
 2165203.7689201477754.2998282312165169.18774818477881.984155302
#Sta/Elev= 30
       0 2944.35    41.8 2940.27    58.8 2931.66    88.5  2914.8   105.5 2906.99
   149.4 2902.07   195.6 2885.36   219.5 2881.63   238.1  2873.6   246.6 2872.69
   276.4 2875.57   294.3 2874.32   324.1 2875.67   327.4 2874.75   332.8 2870.11
   338.2 2868.11   365.2 2867.87     376 2868.59   379.7 2870.08   386.8 2873.21
   392.2 2878.64   397.6 2882.38   413.7 2885.45     425  2895.7   437.3  2909.9
   447.6  2915.6   454.2 2918.45   478.8 2925.13   519.4 2939.43   558.3 2956.18
#Mann= 5 ,-1,0
       0      .1       0  322.61     .06       0   332.8    .045       0
   379.7     .06       0  446.05      .1       0
#XS Ineff= 2 , 0
          320.83 2882.56
Permanent Ineff=
       F       F
Bank Sta=332.8,379.7
XS Rating Curve= 0 ,0
Exp/Cntr(USF)=0,0
Exp/Cntr=0.3,0.1

Type RM Length L Ch R = 1 ,17758   ,404.7,394.7,383.5
XS GIS Cut Line= 3
2164784.80472189477348.6360807672164883.22805734477686.467529475
2164961.70071669477847.402983387
#Sta/Elev= 30
       0 2994.89     4.7 2992.28    21.4 2979.67    54.7 2959.04    67.2 2953.66
      87  2941.5   121.4 2918.98   142.2 2902.95   150.6 2899.55   158.9 2891.77
   177.4 2878.23     188 2868.74   203.2 2858.15   208.9 2855.67   212.9 2855.66
   229.7 2855.77   240.9 2857.83     263 2861.73   275.5 2870.37   279.7 2871.71
   296.4 2870.41   317.2 2872.48   333.9 2878.86   359.3 2893.66   372.7 2899.45
   399.7 2905.93   443.9 2913.34   479.5 2921.66   506.2  2929.7   530.9 2939.84
#Mann= 4 ,-1,0
       0      .1       0   203.2    .045       0   240.9     .06       0
     340      .1       0
Bank Sta=203.2,240.9
XS Rating Curve= 0 ,0
Exp/Cntr(USF)=0,0
Exp/Cntr=0.3,0.1

Type RM Length L Ch R = 1 ,17364   ,461.2,464.8,468.6
XS GIS Cut Line= 2
2164359.19029832477573.4136982142164701.01188225 477928.53573288
#Sta/Elev= 30
       0 2965.44    34.5 2954.79    51.5 2948.28    65.6 2940.41    71.3 2939.71
    77.4 2936.91   105.2 2916.61   116.5 2903.94   127.4 2895.94   151.4 2875.99
   166.2 2861.35   177.3 2845.86   180.2 2844.62   187.2 2844.17   201.4 2844.37
   210.6 2846.13     224 2848.33   238.4 2857.54   252.3 2858.33   278.3 2857.38
   283.4 2858.53   294.7 2863.33   306.1  2864.6   316.1 2867.45   327.2 2869.21
   341.7  2870.6   368.3 2876.75   387.9 2885.85     439 2917.79   492.9 2942.98
#Mann= 5 ,-1,0
       0      .1       0   177.3    .045       0   210.6      .1       0
     230     .06       0     370      .1       0
Bank Sta=177.3,210.6
XS Rating Curve= 0 ,0
Exp/Cntr(USF)=0,0
Exp/Cntr=0.3,0.1

Type RM Length L Ch R = 1 ,16899   ,430.4,433.9,436.7
XS GIS Cut Line= 2
2163994.29371964477793.0578403682164312.02670946478237.884026112
#Sta/Elev= 30
       0 2945.12    39.5 2931.51    84.6 2917.63   104.7  2910.7   120.2 2904.05
   132.9 2901.18   154.6 2891.93   162.4 2889.62     185 2878.76   202.8 2866.14
   226.3 2852.54   236.1 2848.95   255.8 2847.39   262.4 2844.27   275.4 2834.73
   278.5 2833.76   288.2 2831.63     300 2831.12   319.7 2833.36   319.7 2833.38
   344.2 2843.04   381.7  2869.9   398.3 2872.34   411.5 2880.76   429.9 2889.83
   442.6 2894.65   486.8 2918.66   500.4 2924.61     531 2940.75   546.6 2949.72
#Mann= 5 ,-1,0
       0      .1       0   278.5    .045       0   319.7      .1       0
     340     .06       0     460      .1       0
Bank Sta=278.5,319.7
XS Rating Curve= 0 ,0
Exp/Cntr(USF)=0,0
Exp/Cntr=0.3,0.1

Type RM Length L Ch R = 1 ,16465   ,497.9,515.4,533.8
XS GIS Cut Line= 2
2163652.91548407477985.1754621182163938.13626097 478514.23783586
#Sta/Elev= 30
       0 2937.52    54.5 2915.42    81.8 2903.06   104.5 2889.14   116.4 2885.82
   141.2 2865.04   145.4 2863.49   168.1 2862.75   206.1 2835.26   227.2  2832.7
   245.4 2824.59   277.2 2820.42   290.8  2818.8     309 2819.02   322.6 2820.82
   331.7 2824.97     344 2837.05   354.5 2845.01     359 2846.49   372.6 2846.84
   383.3 2853.62   395.1 2864.21   399.9 2866.71   448.2  2888.4     463 2890.65
   477.1 2898.53   492.5 2905.39   537.9 2924.46   563.5 2932.98     601  2949.9
#Mann= 5 ,-1,0
       0      .1       0      90     .06       0   277.2    .045       0
   322.6     .06       0     430      .1       0
Bank Sta=277.2,322.6
XS Rating Curve= 0 ,0
Exp/Cntr(USF)=0,0
Exp/Cntr=0.3,0.1

Type RM Length L Ch R = 1 ,15949   ,374.2,364.8,352.4
XS GIS Cut Line= 3
2163378.66771511478088.4140987062163297.46882697478447.144286205
2163417.27936376478687.802632298
#Sta/Elev= 30
       0 2922.12     9.4 2917.43    29.4 2912.06    47.5 2904.37    74.6 2887.33
    99.2 2885.16   119.6 2871.08   140.2 2861.95     180 2838.87     200 2826.71
     214 2815.82   222.2 2812.37   259.2 2810.84   275.6 2807.46     292  2806.7
   308.4 2805.79   324.8 2806.07   330.5 2807.61   343.8  2815.2   361.7 2821.09
   423.7 2818.91     455    2824   477.3 2835.49   502.6  2853.7   544.4 2879.61
   566.7 2899.18     601 2923.56     610 2926.12   624.8 2924.09   636.6 2931.32
#Mann= 8 ,-1,0
       0     .06       0      80      .1       0     180     .06       0
     200      .1       0     280     .06       0     292    .045       0
   330.5     .06       0  457.81      .1       0
#XS Ineff= 2 , 0
          258.88 2817.96
Permanent Ineff=
       F       F
Bank Sta=292,330.5
XS Rating Curve= 0 ,0
Exp/Cntr(USF)=0,0
Exp/Cntr=0.3,0.1

Type RM Length L Ch R = 1 ,15585   ,441.8,424.1,401.1
XS GIS Cut Line= 3
2162913.80896045478200.024534469 2163017.5524762478674.850625764
2163101.34531584478802.534952835
#Sta/Elev= 30
       0 2912.59    13.5 2911.12    17.6 2909.34    42.1 2888.26    90.3 2849.81
   115.8 2831.14   148.6 2809.83   177.2 2797.02     187 2798.26     218 2797.23
   228.1 2798.23   242.7 2804.59   250.9 2807.02   275.5 2804.98   291.9 2807.37
   310.9 2806.84   336.9 2809.67     382 2808.13   390.1 2809.26   410.6 2809.34
     423 2811.84     470 2814.74   476.1 2816.08   493.6 2823.85   507.9 2833.57
   527.1 2849.53   536.7  2855.4   549.1  2865.1     556 2869.46   638.8 2901.89
#Mann= 6 ,-1,0
       0     .06       0      70      .1       0     187    .045       0
   228.1      .1       0     370     .06       0     470      .1       0
Bank Sta=187,228.1
XS Rating Curve= 0 ,0
Exp/Cntr(USF)=0,0
Exp/Cntr=0.3,0.1

Type RM Length L Ch R = 1 ,15161   ,460.2,482.6,507.2
XS GIS Cut Line= 4
2162436.93845345 478464.422842522162497.89441917478541.831465806
2162813.85992687478754.3992694782162897.93739616 478884.10260497
#Sta/Elev= 30
       0 2860.84    19.9 2854.57    37.6 2851.12    50.5 2846.85    92.6 2837.92
   110.9 2831.33   125.4 2827.38   142.9 2818.25   183.3 2802.31   202.5 2789.63
   229.4 2789.45   260.4 2788.85   274.8 2789.87   289.3 2793.89   305.2 2793.19
   318.7 2796.15     336 2796.24   362.5 2798.74   369.7 2798.65     384 2796.47
   398.3 2799.93     458 2803.18   462.9 2805.07   487.4 2818.55     497 2825.78
   506.2 2834.02   530.3 2851.18   557.1 2865.72   601.3 2881.06   633.9 2896.26
#Mann= 5 ,-1,0
       0      .1       0   229.4    .045       0   274.8      .1       0
  398.53     .06       0  478.53      .1       0
Bank Sta=229.4,274.8
XS Rating Curve= 0 ,0
Exp/Cntr(USF)=0,0
Exp/Cntr=0.3,0.1

Type RM Length L Ch R = 1 ,14678   ,486.4,496.7,509.7
XS GIS Cut Line= 3
 2162297.3464463478494.7814989932162362.89357983 479089.49903549
2162433.67458852479203.912172815
#Sta/Elev= 30
       0  2879.6    14.5  2872.1    82.9 2822.73      95 2815.88   119.1 2798.34
     128 2794.24   149.7 2788.42   171.4 2785.66   191.6 2787.52   204.1 2783.28
   215.7 2786.14   296.2 2790.03   312.3 2786.33   392.8 2785.66   412.9 2781.58
   465.2 2782.15   479.6 2777.97   494.1 2776.97   525.6 2778.28   533.6 2785.69
   541.7 2788.71   566.6  2808.3   581.9 2822.27   607.3 2849.54   628.1 2859.68
   677.5 2892.01   696.7 2908.11   707.2 2914.63   724.9 2928.73   732.9 2932.25
#Mann= 5 ,-1,0
       0      .1       0     460     .06       0   479.6    .045       0
   525.6     .06       0     560      .1       0
#XS Ineff= 2 , 0
          464.58 2794.36
Permanent Ineff=
       F       F
Bank Sta=479.6,525.6
XS Rating Curve= 0 ,0
Exp/Cntr(USF)=0,0
Exp/Cntr=0.3,0.1

Type RM Length L Ch R = 1 ,14181   ,396.9,375.9,356.5
XS GIS Cut Line= 4
 2161891.9909573478571.8501543662161945.19276025478701.899006012
   2161800.36563479108.3016674072161914.15837519479297.463633439
#Sta/Elev= 30
       0 2873.09    14.4 2866.84      36 2859.58    44.7 2853.78    57.6 2849.08
    83.5 2830.85    96.5 2814.45   126.9 2790.67   136.1 2784.69   152.5 2776.52
   165.2 2774.27   194.9 2773.89   250.3 2773.88   296.9 2775.44   309.6  2770.4
   322.3 2767.65   344.2 2766.46   360.6 2763.86   378.7 2766.07   390.3 2767.88
   415.8 2766.74   445.5 2768.49   453.8 2773.42   458.2 2774.37   538.9 2772.23
   555.9 2773.68   607.4 2786.38     671  2804.1   781.1  2862.1   792.7 2866.46
#Mann= 5 ,-1,0
       0      .1       0   344.2    .045       0   378.7      .1       0
  510.51     .06       0  621.95      .1       0
Bank Sta=344.2,378.7
XS Rating Curve= 0 ,0
Exp/Cntr(USF)=0,0
Exp/Cntr=0.3,0.1

Type RM Length L Ch R = 1 ,13805   ,538.3,519,490.3
XS GIS Cut Line= 3
2161402.82993577478765.4456039762161541.34357366479006.160429987
2161858.49813828479294.756850851
#Sta/Elev= 30
       0  2859.5      74 2829.62    82.8 2822.23    93.4 2807.05   112.1 2786.29
   124.3 2774.95   142.8 2762.47   153.1 2759.43   188.3 2760.36   198.1 2756.29
   203.2 2754.22     2382756.343   243.9  2758.5   282.2 2759.22   308.6 2753.59
   317.9 2755.13   330.2 2764.85   338.5 2766.15   373.5 2760.67     413 2764.87
     433 2764.47   454.6 2760.56   484.3 2768.14   502.7 2768.55   519.9 2775.45
   568.2 2775.54   587.7    2783     633 2813.92   656.6 2827.13   706.5 2846.63
#Mann= 5 ,-1,0
       0      .1       0   198.1    .045       0     238      .1       0
  447.72     .06       0  577.72      .1       0
#XS Ineff= 2 , 0
          187.46  2771.8  254.74         2772.06
Permanent Ineff=
       F       F
Bank Sta=198.1,238
XS Rating Curve= 0 ,0
Exp/Cntr(USF)=0,0
Exp/Cntr=0.3,0.1

Type RM Length L Ch R = 1 ,13286   ,363.8,360.5,357
XS GIS Cut Line= 4
2160949.06567087479083.7425023642161041.03890325479257.181506499
2161368.51299116479337.968660748 2161532.4664448479491.703293422
#Sta/Elev= 30
       0 2793.96   119.3 2785.52   164.6 2785.23   194.5 2782.91   207.8 2779.25
   244.9 2759.08   258.4 2754.59   277.8 2752.99     298 2742.88   324.5 2741.32
     341 2741.62   349.82743.135   372.6 2747.14   424.8 2748.75   438.5  2747.5
   475.6 2747.49     493 2742.45   504.4 2741.27   516.8 2745.15   533.3 2748.29
   561.7 2760.99   571.5  2761.5   590.9 2759.41   606.4 2761.38   631.8 2774.93
   653.8  2783.3   672.8 2793.18   699.8 2804.06   725.2 2816.52   758.4 2829.68
#Mann= 5 ,-1,0
       0      .1       0     298    .045       0   349.8      .1       0
  533.61     .06       0  673.61      .1       0
#XS Ineff= 2 , 0
                          400.49         2763.96
Permanent Ineff=
       F       F
Bank Sta=298,349.8
XS Rating Curve= 0 ,0
Exp/Cntr(USF)=0,0
Exp/Cntr=0.3,0.1

Type RM Length L Ch R = 1 ,12926   ,362.7,384.7,401.5
XS GIS Cut Line= 4
2160692.00008137479522.9955323082160831.57271256 479610.02317293
2161312.68778241479667.4942563592161486.74306365 479741.38564934
#Sta/Elev= 30
       0  2832.4    70.9 2805.94    99.2 2793.09   140.2 2757.85   164.3 2742.75
   177.2 2743.99   196.7  2742.1   233.6 2742.55   245.7 2739.02   261.8 2737.35
   338.3  2739.4     355 2735.84   406.8 2735.72   416.32732.629     439 2729.88
   455.1 2731.99   471.2 2734.05   483.3 2739.71   527.6 2739.88   543.8 2736.84
   573.3 2736.79   604.2 2738.88   616.3 2743.76   632.4 2745.25   661.5 2764.79
   704.5 2786.86   722.3 2801.73   753.6 2819.47   799.4 2840.64   838.1 2851.56
#Mann= 5 ,-1,0
       0      .1       0   416.3    .045       0   455.1      .1       0
  614.48     .06       0  709.02      .1       0
#XS Ineff= 2 , 0
          404.76 2749.07
Permanent Ineff=
       F       F
Bank Sta=416.3,455.1
XS Rating Curve= 0 ,0
Exp/Cntr(USF)=0,0
Exp/Cntr=0.3,0.1

Type RM Length L Ch R = 1 ,12541   ,570.9,564.7,555.7
XS GIS Cut Line= 3
2160590.19416215 479613.307234842161097.58172729480145.325264303
2161274.92107044480235.636966835
#Sta/Elev= 30
       0 2846.32    43.4 2824.99      89 2806.01   125.8 2785.51   154.1 2762.67
   182.4 2749.22   202.2 2735.24   215.4 2733.36   228.9 2728.61   306.9 2730.52
   380.4 2726.35   425.4 2728.43   431.8  2726.1   453.1 2724.91   479.4 2722.36
   502.8 2722.94   508.3 2725.12   513.4  2729.1   519.4 2730.68   547.7 2727.24
   609.6  2731.2   624.4 2727.03   640.4 2727.94   697.3 2748.62   727.3 2765.81
   742.9 2772.67     783 2781.22   841.3 2804.91   877.2 2810.25   934.2 2831.74
#Mann= 5 ,-1,0
       0      .1       0     450     .06       0   453.1    .045       0
   508.3     .06       0     580      .1       0
#XS Ineff= 2 ,-1
       0  419.53 2734.49  521.52934.1882 2734.87
Permanent Ineff=
       F       F
Bank Sta=453.1,508.3
XS Rating Curve= 0 ,0
Exp/Cntr(USF)=0,0
Exp/Cntr=0.3,0.1

Type RM Length L Ch R = 1 ,11976   ,412.9,414.3,406.2
XS GIS Cut Line= 5
2160216.47730986480274.2710792232160457.77314012480281.709406179
2160578.07068677480372.9911101152160686.97699413480444.085127882
2160837.96534635480612.322655611
#Sta/Elev= 30
       0 2826.16    41.4 2814.13    75.7 2802.33   131.8 2787.13   155.8 2778.75
   167.8 2772.03   187.8 2755.96   199.8 2747.78   215.8 2734.33     232 2723.99
   249.4 2717.35   269.5 2714.27   309.7 2713.89   331.2  2716.1   388.3 2716.62
   411.4  2712.8   423.6 2715.07   443.2 2714.12   457.7 2711.32   480.8 2711.97
   487.9 2713.98   495.2 2716.69   509.6 2716.78   514.4  2718.5   535.4 2736.12
   555.3 2749.39   608.1 2776.97   626.1 2781.75   685.6 2787.04   748.5  2786.9
#Mann= 5 ,-1,0
       0      .1       0   443.2    .045       0   487.9      .1       0
  492.42     .06       0  632.48      .1       0
#XS Ineff= 2 , 0
          384.93 2756.52
Permanent Ineff=
       F       F
Bank Sta=443.2,487.9
XS Rating Curve= 0 ,0
Exp/Cntr(USF)=0,0
Exp/Cntr=0.3,0.1

Type RM Length L Ch R = 1 ,11562   ,508.9,486.9,445.1
XS GIS Cut Line= 3
2160146.84580427480570.6112816822160560.63760496480823.484048772
2160698.56820519480787.359367759
#Sta/Elev= 30
       0 2816.78    29.7 2806.19    48.4 2794.56   118.8 2757.95   136.7 2745.94
   146.9 2737.54   173.7 2720.04   189.1 2705.61     192 2704.02   198.4 2702.64
   217.2 2702.36   253.1 2703.87   282.8 2707.22   292.2 2706.18     325 2707.49
   337.4 2705.96   353.1 2705.96   360.7 2707.57   369.5 2706.79     386 2709.25
     400 2709.23   427.6 2709.75   456.3 2708.49     480 2709.42   521.7 2708.68
   534.1 2710.92   554.8 2724.82     563 2731.82   596.1 2747.01   627.5 2767.14
#Mann= 7 ,-1,0
       0      .1       0     192    .045       0   253.1      .1       0
     400     .06       0     480      .1       0  504.94     .06       0
  614.94      .1       0
Bank Sta=192,253.1
XS Rating Curve= 0 ,0
Exp/Cntr(USF)=0,0
Exp/Cntr=0.3,0.1

Type RM Length L Ch R = 1 ,11075   ,473.5,452.9,443
XS GIS Cut Line= 5
2160078.73689141481163.9373518232160274.30190931481162.128992052
 2160359.8185326481129.348656154 2160462.0988103481053.681102261
2160752.93603187480943.154757514
#Sta/Elev= 30
       0 2839.42    13.4 2829.24    41.4 2813.08    53.4 2804.18    73.4  2791.7
   125.4 2768.41   160.2  2741.7   181.4 2723.89   189.4 2715.96   201.9 2699.12
   207.12695.037   216.3 2693.79   247.3 2693.46   265.22694.456   274.7 2697.63
   281.4 2698.16   387.6 2694.84     407 2696.92   416.6 2700.59   442.3 2701.03
     468 2704.27   557.8 2703.03   609.2 2704.03   624.2 2708.23   639.1 2716.38
   647.7 2719.58   661.3 2726.52   686.1 2741.89     699 2748.01   725.5 2753.76
#Mann= 5 ,-1,0
       0      .1       0   207.1    .045       0   265.2      .1       0
  544.38     .06       0  654.38      .1       0
#XS Ineff= 2 , 0
                          280.57         2723.74
Permanent Ineff=
       F       F
Bank Sta=207.1,265.2
XS Rating Curve= 0 ,0
Exp/Cntr(USF)=0,0
Exp/Cntr=0.3,0.1

Type RM Length L Ch R = 1 ,10622   ,457.7,487.9,513.8
XS GIS Cut Line= 3
2160147.31889305 481452.717568152160612.90435475481389.343000867
2160817.20403324481205.869958804
#Sta/Elev= 30
       0 2800.94      21 2795.17    73.5 2785.16   105.8 2776.82   170.4 2753.84
   222.9  2740.7     235 2739.24   251.2 2734.32   271.3 2725.72   299.6 2709.34
   319.8 2695.11   327.9 2692.28   360.1 2690.49   380.3 2691.28   392.4 2688.14
   404.6 2687.38   420.7 2689.06   517.6 2687.07   548.7 2683.54   574.3 2680.58
   593.42683.012   603.3 2686.59   613.9 2694.06   625.8 2696.44   643.7 2706.66
   659.3  2713.3   673.4 2722.43   689.3 2729.88   705.5 2733.84   744.5 2746.56
#Mann= 4 ,-1,0
       0      .1       0     440     .06       0   548.7    .045       0
   593.4      .1       0
#XS Ineff= 2 , 0
          517.41 2705.48
Permanent Ineff=
       F       F
Bank Sta=548.7,593.4
XS Rating Curve= 0 ,0
Exp/Cntr(USF)=0,0
Exp/Cntr=0.3,0.1

Type RM Length L Ch R = 1 ,10134   ,324.4,336.1,342.6
XS GIS Cut Line= 3
2160335.20844885481655.2104849442160638.83010003481787.098754632
2160905.86670654 481871.96978989
#Sta/Elev= 30
       0 2729.77      63 2711.63    95.3  2706.9   127.5 2698.73   140.6 2694.04
   153.7 2693.06   158.1 2691.64   166.4 2686.27   171.1  2685.2   187.7 2684.88
   199.9  2680.8   225.8 2677.82   235.9 2678.62   245.5 2681.35   306.3 2682.13
   336.6 2673.47   349.2 2673.45   370.2 2670.62   382.8 2671.22   390.7 2673.53
     407 2677.26   416.4 2682.42   433.2 2683.85   451.6 2698.14   475.1 2707.47
   496.1 2720.94   512.9 2728.96     528 2733.32   575.8 2751.75   611.2 2760.03
#Mann= 4 ,-1,0
       0      .1       0   349.2    .045       0   390.7     .06       0
  481.03      .1       0
Bank Sta=349.2,390.7
XS Rating Curve= 0 ,0
Exp/Cntr(USF)=0,0
Exp/Cntr=0.3,0.1

Type RM Length L Ch R = 1 ,9798    ,428.4,443.6,453.2
XS GIS Cut Line= 2
2160168.62347355481828.7366470432160731.67588806482233.661480578
#Sta/Elev= 30
       0 2756.06    88.1 2730.55   112.8 2721.79   137.4 2704.86   151.9 2698.74
     167 2695.93   186.7 2681.49     192 2679.29   221.2 2677.29   240.5  2672.2
   280.3  2672.4   303.8 2670.32   326.7  2673.5   412.7 2674.31     427 2672.47
   437.9 2666.41   447.1 2664.36   467.5 2662.69   492.9 2664.27     502 2664.81
   507.7 2667.68   521.7 2668.57   535.9 2674.34     556 2676.74     576 2693.22
   590.7  2701.2   610.4 2715.83   620.2 2719.39   639.1 2730.36   693.5 2753.45
#Mann= 5 ,-1,0
       0      .1       0   447.1    .045       0   492.9      .1       0
     510     .06       0     630      .1       0
Bank Sta=447.1,492.9
XS Rating Curve= 0 ,0
Exp/Cntr(USF)=0,0
Exp/Cntr=0.3,0.1

Type RM Length L Ch R = 1 ,9355    ,421.4,416.9,412.4
XS GIS Cut Line= 3
2160151.69333402482213.596735953 2160346.5762987482527.913227736
2160524.96956739482665.345156615
#Sta/Elev= 30
       0 2707.19    18.3 2699.23    38.9 2687.07    49.4 2682.82    65.4 2673.49
    90.1 2661.58   104.6 2661.09   151.1 2663.12   165.6 2662.08   206.6 2661.82
   220.7  2660.5   239.5 2660.79   267.3 2657.43   277.12654.194   281.8 2653.04
   300.7 2651.77   322.5 2651.96     329  2653.4   338.4 2659.11   342.5 2660.65
   352.5 2661.06   357.7 2662.24   374.7  2671.6     392 2682.54   417.5 2695.99
     503 2726.15   511.6 2727.82   538.5  2737.8     562 2745.12     595 2757.29
#Mann= 5 ,-1,0
       0      .1       0     260     .06       0   277.1    .045       0
     329     .06       0     330      .1       0
Bank Sta=277.1,329
XS Rating Curve= 0 ,0
Exp/Cntr(USF)=0,0
Exp/Cntr=0.3,0.1

Type RM Length L Ch R = 1 ,8938    ,501.9,462.1,427.8
XS GIS Cut Line= 3
2159797.24725201482481.1271330842160135.50562876482871.930500406
 2160306.2768481482894.918933778
#Sta/Elev= 30
       0 2746.33    19.1 2744.31    41.1 2729.98    84.7 2710.41   109.9 2697.43
   132.6 2683.44   155.2  2663.7   169.5 2652.85   181.7 2645.41   189.3 2643.32
     217 2643.24   231.8 2645.04   257.3  2651.7   273.4 2652.83   285.7  2655.5
   346.7 2653.77   399.1 2649.76   424.6  2645.6   438.4 2648.25   464.3 2647.24
   475.7 2649.38   499.5 2648.64   511.8 2650.38   521.6  2655.7   561.9 2691.87
   586.1 2709.09   602.3  2715.7   625.3 2722.39   638.6 2728.32   689.2 2739.73
#Mann= 5 ,-1,0
       0      .1       0   181.7    .045       0   231.8      .1       0
     450     .06       0  576.86      .1       0
#XS Ineff= 1 ,-1
  280.83689.1733 2674.96
Permanent Ineff=
       F
Bank Sta=181.7,231.8
XS Rating Curve= 0 ,0
Exp/Cntr(USF)=0,0
Exp/Cntr=0.3,0.1

Type RM Length L Ch R = 1 ,8476    ,423.7,444.6,457.3
XS GIS Cut Line= 4
2159739.32283667483087.0365555292159849.79224257483072.258276932
2160107.59110253482972.0943886692160280.00435282482977.020481535
#Sta/Elev= 30
       0  2683.6     4.9 2682.32      17 2676.44    37.2 2668.18    81.6 2657.94
   109.8 2645.66   126.9 2642.51   139.8 2634.55   146.6  2633.3   161.2 2633.01
   191.3 2634.03   199.8 2636.75   208.4  2638.5     217 2639.14   234.2 2643.74
   285.7 2642.41   302.8 2640.65   315.7 2641.74   371.5 2642.33   375.8 2642.98
     388 2648.55   392.6 2651.65   420.6 2675.65   452.6 2699.79   464.6 2706.59
   484.7 2713.02   504.7 2716.73   541.4 2731.73   552.7 2735.94   560.5 2737.86
#Mann= 5 ,-1,0
       0      .1       0   139.8    .045       0   191.3      .1       0
  261.45     .06       0  468.03      .1       0
Bank Sta=139.8,191.3
XS Rating Curve= 0 ,0
Exp/Cntr(USF)=0,0
Exp/Cntr=0.3,0.1

Type RM Length L Ch R = 1 ,8031    ,257.6,256.6,254.4
XS GIS Cut Line= 3
2159622.75861994483310.8618436762160171.19695895483519.399774978
2160315.69568301483514.473682112
#Sta/Elev= 30
       0 2697.69    35.8  2682.1    48.6 2680.14    74.3 2667.38   104.2  2657.6
   121.3 2647.35   138.5 2634.51     147 2630.53   204.4 2628.39     284  2630.5
   313.9  2632.6   343.9 2629.62   365.3 2624.39   399.8 2624.98   420.9 2622.99
   429.5  2623.2   433.5  2624.8   449.4 2633.26     468 2634.09   481.8 2636.73
   493.6 2643.63   511.4 2659.31     545 2677.28   628.5 2711.81   667.8  2726.6
   687.8 2736.12   695.8 2737.82   707.8 2745.42   723.8  2750.2   731.3  2753.9
#Mann= 5 ,-1,0
       0      .1       0   399.8    .045       0   433.5      .1       0
     470     .06       0  606.75      .1       0
#XS Ineff= 2 , 0
          309.68 2644.49
Permanent Ineff=
       F       F
Bank Sta=399.8,433.5
XS Rating Curve= 0 ,0
Exp/Cntr(USF)=0,0
Exp/Cntr=0.3,0.1

Type RM Length L Ch R = 1 ,7775    ,293,296,298.5
XS GIS Cut Line= 3
2159512.74254595483560.4505488562160103.87368979483750.926139652
2160241.80429003483739.431922966
#Sta/Elev= 30
       0 2699.24    58.2 2679.57    96.1 2671.79   108.7 2668.03   125.5 2659.13
   142.3 2646.29   154.9 2638.36   171.9 2625.14   181.3 2620.56   286.2  2624.4
   318.8 2623.45   352.4 2625.51   381.8 2624.84     386 2624.28   394.4 2620.89
   410.1 2618.29   435.6 2617.27   457.5  2617.5     463 2618.54   465.9  2619.5
   478.5 2627.81   499.5  2631.6   507.9 2637.85   512.1 2639.89   541.5 2646.82
   570.9 2657.06   629.4 2674.73   689.5 2698.72   721.7 2707.47   759.5 2720.05
#Mann= 5 ,-1,0
       0      .1       0     400     .06       0   410.1    .045       0
     463     .06       0     610      .1       0
#XS Ineff= 2 , 0
          371.07 2653.18
Permanent Ineff=
       F       F
Bank Sta=410.1,463
XS Rating Curve= 0 ,0
Exp/Cntr(USF)=0,0
Exp/Cntr=0.3,0.1

Type RM Length L Ch R = 1 ,7479    ,133.3,138.1,142
XS GIS Cut Line= 3
2159455.27146252483816.6073778572159954.44887288484025.145309159
2160172.83898991483989.020628146
#Sta/Elev= 30
       0 2688.99    62.3 2665.76    74.7 2655.68    83.7 2650.65    96.3 2637.02
     105 2629.52   122.4 2618.94     131 2616.33   152.7 2612.92   161.4 2615.74
   250.5 2616.29   287.1  2619.6   321.8 2617.81   339.1 2620.43   364.7 2616.85
   374.2 2613.98   382.5 2611.57   395.2 2610.79   421.5 2611.25   430.1 2614.05
   441.4 2625.04   447.5 2627.97   468.9 2627.33   482.2  2629.4   538.5 2628.72
   554.9 2640.39     563 2643.93   611.7 2653.76   684.6 2673.45   762.3 2691.46
#Mann= 5 ,-1,0
       0      .1       0   374.2    .045       0   430.1      .1       0
     480     .06       0  680.99      .1       0
#XS Ineff= 2 , 0
          340.35 2633.09
Permanent Ineff=
       F       F
Bank Sta=374.2,430.1
XS Rating Curve= 0 ,0
Exp/Cntr(USF)=0,0
Exp/Cntr=0.3,0.1

Type RM Length L Ch R = 1 ,7340    ,436,455.5,464.1
XS GIS Cut Line= 3
2159424.07287437483897.0668946582159885.48357276 484163.07590939
2159997.14167771484414.306645526
#Sta/Elev= 30
       0 2695.37    40.3 2679.24    52.9 2671.59    78.6 2651.36    87.8 2638.42
   104.3 2623.87   115.5 2615.15   124.8 2611.06   155.4 2613.44   166.3 2612.27
   176.4 2614.15     214 2612.72   296.5 2614.69   304.8 2614.36   323.3 2610.28
   351.6 2610.85   368.6 2609.81   401.8 2611.06   424.8 2623.21   440.7 2627.73
     508  2632.6   539.3 2631.75   554.4 2634.52   648.4 2637.16   663.5 2639.59
     687 2639.42   718.7 2643.07   758.1  2642.9   793.2 2648.88   807.5 2648.84
#Mann= 5 ,-1,0
       0      .1       0   351.6    .045       0   401.8      .1       0
   542.6     .06       0   652.6      .1       0
#XS Ineff= 2 , 0
          301.05 2621.86
Permanent Ineff=
       F       F
Bank Sta=351.6,401.8
XS Rating Curve= 0 ,0
Exp/Cntr(USF)=0,0
Exp/Cntr=0.3,0.1

Type RM Length L Ch R = 1 ,6885    ,486,488.8,489
XS GIS Cut Line= 4
2159181.86788135484042.5593511882159428.52242035484392.322811682
2159536.68251209484460.4236101872159597.11222659 484680.43261879
#Sta/Elev= 30
       0 2730.07    32.6 2716.71    47.3 2707.93    76.6 2697.96   140.3 2672.64
   175.8 2650.47   228.4 2608.72     240 2606.62   250.3 2602.78   270.2 2602.58
   284.8 2601.38   305.72602.328   316.5 2605.57   362.3  2606.9   385.3 2610.16
   420.4 2608.57   428.4 2610.72   444.6 2619.32   459.6 2621.74   474.6 2622.19
   518.3 2619.57   553.1 2621.38     569 2628.16   598.1 2630.48   656.1 2644.85
   673.2 2650.84   705.9 2666.41     735  2676.2   751.5 2679.77     784  2683.5
#Mann= 5 ,-1,0
       0      .1       0   270.2    .045       0   305.7      .1       0
  517.99     .06       0   665.8      .1       0
Bank Sta=270.2,305.7
XS Rating Curve= 0 ,0
Exp/Cntr(USF)=0,0
Exp/Cntr=0.3,0.1

Type RM Length L Ch R = 1 ,6396    ,318.1,330.4,344.5
XS GIS Cut Line= 4
 2158821.8226964484199.6288225772158924.36048472484498.579778581
 2159171.1414613484798.9246380462159198.48398554484878.168544134
#Sta/Elev= 30
       0 2708.49    56.6  2686.4    94.4 2658.46   111.6 2647.42   149.6 2613.92
   162.3 2606.14     175  2602.5   204.7 2598.35   229.2 2599.56   242.7 2598.17
   276.5 2598.48   305.4 2601.87   328.4 2601.08   351.9 2597.79   391.4 2599.33
   467.82596.396     494 2593.75   516.1 2593.63   528.1 2596.14   536.6  2599.7
     565 2601.58   580.4 2607.54   616.2 2608.07   640.4 2603.54   697.3 2606.35
   707.2 2611.52   724.1 2625.06   745.2 2639.52   762.2 2642.12   788.6 2640.62
#Mann= 5 ,-1,0
       0      .1       0   467.8    .045       0   528.1      .1       0
  606.05     .06       0  774.77      .1       0
#XS Ineff= 2 , 0
          412.57 2615.62
Permanent Ineff=
       F       F
Bank Sta=467.8,528.1
XS Rating Curve= 0 ,0
Exp/Cntr(USF)=0,0
Exp/Cntr=0.3,0.1

Type RM Length L Ch R = 1 ,6066    ,293.3,305.7,339.4
XS GIS Cut Line= 3
 2158559.7482939484387.0186475892158653.34405834 484511.81300018
2158840.53558723485040.546967733
#Sta/Elev= 30
       0 2692.16      14 2685.96    37.7 2678.09    47.7 2672.29    67.6 2656.56
    77.7 2646.66    93.3 2635.21     114 2617.47   144.7 2597.26   153.3 2593.22
   199.9 2592.62   258.7 2594.19   280.5 2591.57   344.2 2590.34   361.1 2592.51
   390.8 2592.74   416.3 2592.13   420.5 2590.72   433.3 2589.16   496.9 2590.82
   505.4 2595.17   509.6 2596.03   522.4 2596.67   539.3 2599.46   581.8 2601.03
   598.7  2605.5   624.2 2606.54   657.6 2620.71   687.9 2636.94   716.9  2641.4
#Mann= 5 ,-1,0
       0      .1       0   420.5    .045       0   496.9      .1       0
  525.99     .06       0  625.99      .1       0
#XS Ineff= 2 , 0
          259.65  2604.3
Permanent Ineff=
       F       F
Bank Sta=420.5,496.9
XS Rating Curve= 0 ,0
Exp/Cntr(USF)=0,0
Exp/Cntr=0.3,0.1

Type RM Length L Ch R = 1 ,5760    ,218.3,193.2,177.8
XS GIS Cut Line= 3
2158519.07672097484394.5982248562158448.07162371484771.188964035
2158545.78291646485013.291753751
#Sta/Elev= 30
       0 2690.86    39.3 2672.67   100.6 2626.86   120.7 2615.41   145.1 2596.93
   153.2 2592.54   161.4 2590.35   193.9  2590.3   218.4 2587.58   242.8 2589.16
   258.1 2587.19   282.1 2581.57   307.9 2579.65   332.3 2579.83   345.7 2581.84
   356.8 2586.34     378 2586.37   398.3 2595.84   411.3  2597.5   419.9 2602.31
   426.3 2603.64   467.8  2606.5   501.1 2610.53   579.5 2623.43   596.7 2628.55
     601 2628.47   609.7 2624.16   615.3 2623.81   631.2 2631.39   644.3 2632.63
#Mann= 4 ,-1,0
       0      .1       0   282.1    .045       0   345.7      .1       0
  563.23     .06       0
Bank Sta=282.1,345.7
XS Rating Curve= 0 ,0
Exp/Cntr(USF)=0,0
Exp/Cntr=0.3,0.1

Type RM Length L Ch R = 1 ,5567    ,266.9,259.2,256.2
XS GIS Cut Line= 3
2158234.37585986484373.4629775722158251.18019744484657.131254122
2158411.23363883 485045.56238074
#Sta/Elev= 30
       0 2671.41    55.8 2641.18    83.9 2623.29    95.9 2613.21   107.9 2606.57
   127.9 2590.63     140 2584.13     148 2582.99     160 2584.22   243.5 2585.22
   264.2 2582.34   291.1 2584.35   297.3 2582.84   304.5 2578.79   318.7 2576.82
   357.8 2577.51   366.4 2579.05     388 2578.54   405.4 2581.47   448.6 2582.37
   453.5 2584.18   474.9 2598.43   487.6  2603.1   539.5 2606.55   595.7 2612.32
     625 2617.37   669.3 2623.17   683.3 2625.83   695.2  2629.9   704.3 2630.72
#Mann= 3 ,-1,0
       0      .1       0   304.5    .045       0   366.4      .1       0
#XS Ineff= 2 , 0
          289.97 2595.79   417.3         2595.79
Permanent Ineff=
       F       F
Bank Sta=304.5,366.4
XS Rating Curve= 0 ,0
Exp/Cntr(USF)=0,0
Exp/Cntr=0.3,0.1

Type RM Length L Ch R = 1 ,5308    ,424.3,437.1,449.4
XS GIS Cut Line= 2
2157843.82279746484455.9839477052158183.72320517485089.807896387
#Sta/Elev= 30
       0 2632.86    33.1  2612.5    66.1 2595.15    92.1 2585.39   128.4 2578.86
   155.7 2575.79   187.4 2577.69   232.8 2576.61   260.1 2578.66   314.5 2578.29
   359.9 2580.53   391.7 2578.15   405.3 2578.36   432.7 2570.73   450.7 2568.51
   468.9 2570.24   482.5 2570.38   497.5 2572.33   506.4 2575.81   518.8 2577.47
   527.9 2581.72   550.7 2597.67   555.1 2599.47   614.1 2612.39   632.3 2617.44
   648.2 2623.24     664 2626.46   691.3 2634.79   713.2 2639.54   719.2 2641.69
#Mann= 4 ,-1,0
       0      .1       0   432.7    .045       0   468.9      .1       0
     680     .06       0
Bank Sta=432.7,468.9
XS Rating Curve= 0 ,0
Exp/Cntr(USF)=0,0
Exp/Cntr=0.3,0.1

Type RM Length L Ch R = 1 ,4871    ,475.4,470.8,469.6
XS GIS Cut Line= 3
2157638.21632063484468.0292537722157630.82718133484639.457285488
2157652.99459922485162.608347794
#Sta/Elev= 30
       0 2671.41    37.6 2650.32    77.2 2633.02   125.9 2609.83   141.3 2599.54
   165.3 2580.98   185.3 2570.06   189.3 2569.01   201.3 2567.53   209.3 2569.64
   261.4  2571.1   325.4 2569.38   341.5 2572.43   381.5 2572.44     405 2570.34
   417.5  2565.7   457.6 2567.67   489.5 2565.64   504.8 2561.77   541.6 2560.87
   554.8 2561.42   557.7 2562.34   565.7 2568.18   581.7 2570.43   589.7 2575.82
   600.9 2579.53   609.7 2586.93   617.7 2590.63   658.5 2600.06   695.2 2611.95
#Mann= 3 ,-1,0
       0      .1       0   504.8    .045       0   554.8      .1       0
#XS Ineff= 2 , 0
          451.73 2585.21
Permanent Ineff=
       F       F
Bank Sta=504.8,554.8
XS Rating Curve= 0 ,0
Exp/Cntr(USF)=0,0
Exp/Cntr=0.3,0.1

Type RM Length L Ch R = 1 ,4400    ,510.4,485.9,467.8
XS GIS Cut Line= 4
2157174.18183206484682.6442651252157174.51180377484876.903117503
2157220.66522028485163.9720924382157395.48748194485307.765449745
#Sta/Elev= 30
       0 2632.61    66.5 2607.43    90.5 2595.75   138.5 2577.28   162.5 2563.38
   182.5 2561.14   199.4 2556.46   214.8  2556.2   220.4 2554.11   226.9 2552.19
   255.1 2551.94   267.5 2553.69   287.7 2554.51   299.9 2557.47   324.2  2557.9
   340.4 2557.08   349.5 2554.01   356.6 2553.51     389 2560.52   401.9 2558.75
   482.2  2558.5   499.7 2556.52   524.7 2560.14   567.9 2559.56   581.4 2564.37
   599.2 2577.26   606.6 2580.56   631.7 2588.26   653.2 2592.33   711.4 2608.38
#Mann= 6 ,-1,0
       0      .1       0   220.4    .045       0   267.5      .1       0
  474.26     .06       0  625.01      .1       0  635.01     .06       0
#XS Ineff= 2 , 0
                          389.13         2572.77
Permanent Ineff=
       F       F
Bank Sta=220.4,267.5
XS Rating Curve= 0 ,0
Exp/Cntr(USF)=0,0
Exp/Cntr=0.3,0.1

Type RM Length L Ch R = 1 ,3914    ,468.6,465.8,463
XS GIS Cut Line= 3
2156717.52956408485088.7169548132156770.73136703485208.421011442
2157184.52316772485524.676173401
#Sta/Elev= 30
       0 2583.83    26.2 2579.86    36.1 2579.46    95.2 2568.24   118.7 2562.33
   135.4 2554.84   145.4 2551.55   181.1  2547.7   204.7 2543.43   211.3 2543.42
   243.6 2542.36   253.6 2543.71   263.7 2550.62   293.9 2550.57   332.3 2554.32
   354.3 2552.45   389.6 2551.56   403.7 2552.42   422.1 2555.68   475.2 2554.62
   480.7 2556.01   490.3 2561.82   495.3 2563.74   505.4  2564.7   526.4 2564.29
   547.2 2568.38   573.6 2579.29   586.3 2582.11   623.4 2598.03   651.8 2608.79
#Mann= 5 ,-1,0
       0      .1       0   211.3    .045       0   253.6      .1       0
  360.99     .06       0  530.99      .1       0
Bank Sta=211.3,253.6
XS Rating Curve= 0 ,0
Exp/Cntr(USF)=0,0
Exp/Cntr=0.3,0.1

Type RM Length L Ch R = 1 ,3448    ,448.6,456.1,464.2
XS GIS Cut Line= 3
2156381.80518571485393.6319671872156482.15152186485585.202245286
2156863.46759922485827.857930878
#Sta/Elev= 30
       0 2582.72    62.7 2573.94    71.7 2570.53    85.3 2563.66   116.9 2551.76
   130.4 2547.34     144 2544.68   180.1 2542.65   202.9 2544.16   217.7 2542.14
   228.1 2539.22   247.1 2540.96   272.8 2541.75   290.1 2538.89   301.7 2538.72
   335.4 2538.52   359.7  2538.8   368.4 2540.08   380.1 2544.19   487.2 2543.19
   521.7 2544.39   526.8 2546.53   542.2 2557.13   562.5 2567.47     577 2576.71
   603.6 2590.69   626.2  2604.9   640.6 2610.75   658.1 2615.61   668.2  2619.7
#Mann= 5 ,-1,0
       0      .1       0  296.26     .06       0   301.7    .045       0
   359.7     .06       0  516.26      .1       0
#XS Ineff= 2 , 0
          204.07 2552.77  379.94         2556.78
Permanent Ineff=
       F       F
Bank Sta=301.7,359.7
XS Rating Curve= 0 ,0
Exp/Cntr(USF)=0,0
Exp/Cntr=0.3,0.1

Type RM Length L Ch R = 1 ,2992    ,459.9,462.8,468.7
XS GIS Cut Line= 3
2156092.17101315485453.4811481772156179.74599742485867.637844639
2156572.00894782486292.741414135
#Sta/Elev= 30
       0 2590.93    69.2 2567.94     106 2549.41   130.5 2540.01     200 2540.58
   216.4 2536.46   240.9  2534.6   265.4 2537.92   326.8 2533.82   343.1 2537.49
   430.4 2539.21   447.5 2532.32   458.7 2530.53   471.1 2533.79   560.6 2534.65
   586.1 2534.06     605 2530.59   632.2 2528.33   654.3 2530.43   662.5  2535.5
   736.1 2534.11   744.6 2536.03   762.9 2549.09   789.6 2579.72   801.4  2587.6
   833.6 2604.12     888  2626.1   915.3 2640.49   960.7 2667.43  1001.7 2694.57
#Mann= 5 ,-1,0
       0      .1       0     605    .045       0   654.3      .1       0
  663.31     .06       0  793.31      .1       0
#XS Ineff= 2 , 0
          428.21 2548.12  675.42         2544.81
Permanent Ineff=
       F       F
Bank Sta=605,654.3
XS Rating Curve= 0 ,0
Exp/Cntr(USF)=0,0
Exp/Cntr=0.3,0.1

Type RM Length L Ch R = 1 ,2529    ,490,495.3,499.6
XS GIS Cut Line= 3
2155601.38620545 485504.56655567  2155776.536174486046.436770864
2156176.09703975486590.131464898
#Sta/Elev= 30
       0 2614.09    17.5 2604.11    80.5 2577.03   113.1 2558.28   148.8 2531.84
   160.4 2526.79   261.3 2529.31   315.9 2525.17   353.8 2528.42     421 2526.93
   454.7 2530.43   507.8 2527.04   568.3 2531.38   647.3  2526.1   702.8 2527.82
     720 2524.18     758 2523.69   781.4 2528.49   885.6 2523.22   930.3 2523.49
   979.9 2521.49   989.9 2523.58  1021.4 2542.98  1034.7 2555.88  1046.1 2572.74
  1054.7 2579.09  1129.1  2600.7  1193.4 2640.11  1223.2 2649.06  1244.2  2661.3
#Mann= 6 ,-1,0
       0      .1       0  869.47     .08       0  929.47     .06       0
   930.3    .045       0   989.9     .06       0 1049.47      .1       0
#XS Ineff= 2 , 0
          696.77 2548.29
Permanent Ineff=
       F       F
Bank Sta=930.3,989.9
XS Rating Curve= 0 ,0
Exp/Cntr(USF)=0,0
Exp/Cntr=0.3,0.1

Type RM Length L Ch R = 1 ,2034    ,473.7,483.5,478.9
XS GIS Cut Line= 4
2155279.14392205 485607.169227942155453.13541188486338.170408876
2155639.63769321486699.0117792632155726.80723774486782.126926375
#Sta/Elev= 30
       0 2626.17    10.3 2620.22    18.5 2619.54    26.7 2615.51   100.7 2562.45
   158.3 2537.88   178.9 2523.13   187.1 2520.15     294 2520.97   335.1 2519.22
   450.2 2523.06   511.9 2520.01   614.7 2520.97   643.5 2517.47   684.6 2521.25
   810.3 2517.19   853.9 2520.25   868.7 2514.41   919.2 2518.95   939.4 2517.71
   952.9  2514.3   970.9 2518.71  1002.5 2519.41  1054.2 2515.69  1097.3 2515.53
  1118.1 2517.69  1128.5 2525.64    1142 2527.26  1166.5  2545.6  1278.1 2587.35
#Mann= 4 ,-1,0
       0      .1       0  1054.2    .045       0  1097.3     .06       0
 1197.61      .1       0
#XS Ineff= 2 , 0
          854.32 2539.12
Permanent Ineff=
       F       F
Bank Sta=1054.2,1097.3
XS Rating Curve= 0 ,0
Exp/Cntr(USF)=0,0
Exp/Cntr=0.3,0.1

Type RM Length L Ch R = 1 ,1550    ,401.8,413.9,401.6
XS GIS Cut Line= 3
2154896.95558631485755.6469238072155196.55553394486925.841122393
 2155157.1127541487151.786183557
#Sta/Elev= 30
       0 2611.63    22.2 2592.23   117.2 2522.32   128.8 2515.61     142 2510.94
   222.6 2512.32   265.8 2508.02   294.7 2511.22   377.3  2513.8   435.1 2510.59
   468.2 2514.52   529.1 2514.23   596.2 2518.33   612.1 2517.76   633.3 2512.23
   691.1    2513   765.4 2508.53   794.4  2510.1   810.9 2507.33     910 2512.12
   921.1 2508.53   930.6 2506.06   946.7    2506   990.1 2506.28   999.72508.112
  1087.5 2516.41  1124.3 2516.83  1182.5  2533.2  1363.3 2541.03  1437.3 2562.46
#Mann= 5 ,-1,0
       0      .1       0   921.1    .045       0   999.7      .1       0
    1110     .06       0 1207.94      .1       0
#XS Ineff= 2 , 0
          596.71 2537.87
Permanent Ineff=
       F       F
Bank Sta=921.1,999.7
XS Rating Curve= 0 ,0
Exp/Cntr(USF)=0,0
Exp/Cntr=0.3,0.1
